--- wekiva_ras.prj (project) ---

Proj Title=wekiva_ras
Current Plan=p01
Default Exp/Contr=0.3,0.1
English Units
Geom File=g05
Geom File=g01
Flow File=f03
Unsteady File=u01
Unsteady File=u02
Plan File=p03
Plan File=p01
Y Axis Title=Elevation
X Axis Title(PF)=Main Channel Distance
X Axis Title(XS)=Station
BEGIN DESCRIPTION:
END DESCRIPTION:
DSS File=dss
DSS Export Rating Curves= 0
DSS Export Rating Curve Sorted= 0
DSS Export Volume Flow Curves= 0
DXF OffsetX= 0
DXF OffsetY= 0
DXF ScaleX= 1
DXF ScaleY= 10
Specific Locations Profile Table=stations                             , 8
LtWekiva        ,LtWekiva        ,312.14
LtWekiva        ,LtWekiva        ,248.51
ROK             ,ROK             ,480.77
ROK             ,ROK             ,126.88
wekiva          ,wek_run         ,793.32
wekiva          ,wekiva_riv_up   ,739.30
wekiva          ,wekiva_riv_down ,405.81
wekiva          ,wekiva_riv_down ,318.86

--- wekiva_ras.p01 (plan) ---

Plan Title=unsteady_2009
Program Version=5.03
Short Identifier=U2009
Simulation Date=20JAN2009,2400,20JUL2009,2300
Geom File=g01
Flow File=u02
Subcritical Flow
K Sum by GR= 0
Std Step Tol= 0.01
Critical Tol= 0.01
Num of Std Step Trials= 20
Max Error Tol= 0.3
Flow Tol Ratio= 0.001
Split Flow NTrial= 30
Split Flow Tol= 0.02
Split Flow Ratio= 0.02
Log Output Level= 0
Friction Slope Method= 1
Unsteady Friction Slope Method= 2
Unsteady Bridges Friction Slope Method= 1
Parabolic Critical Depth
Global Vel Dist= 0 , 0 , 0
Global Log Level= 0
CheckData=True
Encroach Param=-1 ,0,0, 0
Computation Interval=30MIN
Output Interval=1DAY
Instantaneous Interval=1DAY
Mapping Interval=1DAY
Run HTab= 1
Run UNet= 1
Run Sediment= 0
Run PostProcess= 1
Run WQNet= 0
Run RASMapper= 0
UNET Theta= 1
UNET Theta Warmup= 1
UNET ZTol= 0.02
UNET ZSATol= 0.02
UNET MxIter= 20
UNET Max Iter WO Improvement= 0
UNET MaxInSteps= 0
UNET DtIC= 0
UNET DtMin= 0
UNET MaxCRTS= 20
UNET WFStab= 2
UNET SFStab= 1
UNET WFX= 1
UNET SFX= 1
UNET DSS MLevel= 4
UNET Pardiso=0
UNET DZMax Abort= 100
UNET Use Existing IB Tables=-1
UNET Froude Reduction=True
UNET Froude Limit= 0.8
UNET Froude Power= 4
UNET Time Slicing=0,0, 5
UNET D1 Cores= 0
UNET D2 Coriolis=0
UNET D2 Cores= 0
UNET D2 Theta= 1
UNET D2 Theta Warmup= 1
UNET D2 Z Tol= 0.01
UNET D2 Volume Tol= 0.01
UNET D2 Max Iterations= 20
UNET D2 Equation= 0
UNET D2 RampUpFraction=0.1
UNET D2 TimeSlices= 1
UNET D2 BCVolumeCheck=0
UNET D1D2 MaxIter= 0
UNET D1D2 ZTol=0.01
UNET D1D2 QTol=0.1
UNET D1D2 MinQTol=1
DSS File=dss
Write IC File= 0
Write IC File at Fixed DateTime=0
Write IC File at Sim End=0
Echo Input=False
Echo Parameters=False
Echo Output=False
Write Detailed= 0
HDF Write Warmup=0
HDF Write Time Slices=0
HDF Flush=0
HDF Face Node Velocities=0
HDF Compression= 1
HDF Chunk Size= 1
HDF Spatial Parts= 1
HDF Use Max Rows=0
HDF Fixed Rows= 1
Calibration Method= 0
Calibration Iterations= 20
Calibration Max Change=0.05
Calibration Tolerance=0.2
Calibration Maximum=1.5
Calibration Minimum=0.5
Calibration Optimization Method= 1
WQ AD Non Conservative
WQ ULTIMATE=-1
WQ Max Comp Step=1HOUR
WQ Output Interval=15MIN
WQ Output Selected Increments= 0
WQ Output face flow=0
WQ Output face velocity=0
WQ Output face area=0
WQ Output face dispersion=0
WQ Output cell volume=0
WQ Output cell surface area=0
WQ Output cell continuity=0
WQ Output cumulative cell continuity=0
WQ Output face conc=0
WQ Output face dconc_dx=0
WQ Output face courant=0
WQ Output face peclet=0
WQ Output face adv mass=0
WQ Output face disp mass=0
WQ Output cell mass=0
WQ Output cell source sink temp=0
WQ Output nsm pathways=0
WQ Output nsm derived pathways=0
WQ Output MaxMinRange=-1
WQ Daily Max Min Mean=-1
WQ Daily Range=0
WQ Daily Time=0
WQ Create Restart=0
WQ Fixed Restart=0
WQ System Summary=0
WQ Write To DSS=0
WQ Use Fixed Temperature=0
Sorting and Armoring Iterations= 10
XS Update Threshold= 0.02
Bed Roughness Predictor= 0
Hydraulics Update Threshold= 0.02
Energy Slope Method= 1
Volume Change Method= 1
Sediment Retention Method= 0
XS Weighting Method= 0
Number of US Weighted Cross Sections= 1
Number of DS Weighted Cross Sections= 1
Upstream XS Weight=0
Main XS Weight=1
Downstream XS Weight=0
Number of DS XS's Weighted with US Boundary= 1
Upstream Boundary Weight= 1
Weight of XSs Associated with US Boundary= 0
Number of US XS's Weighted with DS Boundary= 1
Downstream Boundary Weight= 0.5
Weight of XSs Associated with DS Boundary= 0.5
Percentile Method= 0
Sediment Output Level= 4
Mass or Volume Output= 0
Output Increment Type= 1
Profile and TS Output Increment= 1
XS Output Flag= 0
XS Output Increment= 10
Write Gradation File= 0
Read Gradation Hotstart= 0
Write HDF5 File= 1
Write DSS Sediment File= 0
SV Curve= 0
Specific Gage Flag= 0

--- wekiva_ras.p03 (plan) ---

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Plan Title=Plan 03
Short Identifier=Plan 03
Simulation Date=01JUN2008,2400,31OCT2008,2300
Geom File=g01
Flow File=u01
Computation Interval=1HOUR

--- wekiva_ras.f03 (steady flow) ---

Flow Title=Flow 03
Program Version=5.03
Number of Profiles= 14
Profile Names=PF 1,PF 2,PF 3,PF 4,PF 5,PF 6,PF 7,PF 8,PF 9,PF 10,PF 11,PF 12,PF 13,PF 14
River Rch & RM=LtWekiva,LtWekiva        ,312.14
     .87    44.8     279     269     536     340     269     295    64.8    80.3
    20.5    14.1    5.33      .4
River Rch & RM=LtWekiva,LtWekiva        ,245.69
   29.12   99.89  320.24  327.25  576.71  382.65  327.25  345.13  112.27  113.58
   57.32   47.52   35.97   29.47
River Rch & RM=LtWekiva,LtWekiva        ,182.49
   29.34  118.51  326.64  333.11     640  398.61  333.11  354.77  113.77  114.81
   58.05   47.94   36.21   29.67
River Rch & RM=LtWekiva,LtWekiva        ,30.50
   29.09  140.12  319.54  448.57  1020.7  433.21  448.57  384.36  140.02  216.28
   62.67   51.63   34.72   30.07
River Rch & RM=ROK,ROK             ,480.77
   46.81   50.62   58.99    59.1    72.3    56.8    59.1   59.07   58.21   56.78
   56.06   48.82   48.07   45.98
River Rch & RM=ROK,ROK             ,350.27
   46.81   53.87   66.43   65.06  118.02   69.39   65.06   65.39   61.15   60.37
   58.17   49.14   48.14   45.98
River Rch & RM=ROK,ROK             ,215.81
   48.06   60.87   72.93   72.45  244.78   79.49   72.45   73.43   68.89   71.45
   67.01   50.91   50.04   47.05
River Rch & RM=ROK,ROK             ,18.17
   52.63  118.28  135.41   184.5  421.87  173.02   184.5  162.67  119.14   84.39
    72.6   58.73   56.24   54.45
River Rch & RM=wekiva,wek_run         ,793.32
   50.49   59.48   58.93   59.35      58    57.3   59.35   59.98   54.97   65.09
    63.3   54.43   52.19   50.23
River Rch & RM=wekiva,wekiva_riv_up   ,747.19
  103.56   187.4  196.33  246.07  529.08  237.32  246.07  227.83  176.25  151.98
  137.87  113.83  108.94  105.06
River Rch & RM=wekiva,wekiva_riv_up   ,579.74
  109.22  260.39  254.11  363.38  546.77  348.55  363.38  311.47  274.16  196.47
  136.52  120.89  116.29   114.1
River Rch & RM=wekiva,wekiva_riv_down ,544.57
  138.31   400.5  573.65  811.95 1567.47  781.77  811.95  695.84  414.18  412.75
   199.2  172.52  151.01  144.17
River Rch & RM=wekiva,wekiva_riv_down ,477.90
  134.46  381.67     644  897.74 1712.97   900.7  897.74  771.58  456.61  451.02
  210.91  180.44  147.97  139.01
River Rch & RM=wekiva,wekiva_riv_down ,386.11
  149.45  398.62  662.25  915.94 1732.87  919.32  915.94  789.81  473.88  469.05
  226.53  196.41  163.38  153.51
River Rch & RM=wekiva,wekiva_riv_down ,333.01
     150     407     665     927    1740     922     927     797     479     467
     225     196     164     155
River Rch & RM=wekiva,wekiva_riv_down ,143.23
  164.13  395.45  662.21  992.42 1896.43   896.8  992.42     837  552.92   520.6
   259.2  235.86  178.61  169.47
River Rch & RM=wekiva,wekiva_riv_down ,25.630*
   192.3  496.71  976.34 1309.67 3142.04 1327.24 1309.67 1149.23  674.13  799.64
  336.48  291.63  213.14  196.75
Boundary for River Rch & Prof#=LtWekiva,LtWekiva        , 1
Up Type= 0
Dn Type= 0
Boundary for River Rch & Prof#=LtWekiva,LtWekiva        , 2
Up Type= 0
Dn Type= 0
Boundary for River Rch & Prof#=LtWekiva,LtWekiva        , 3
Up Type= 0
Dn Type= 0
Boundary for River Rch & Prof#=LtWekiva,LtWekiva        , 4
Up Type= 0
Dn Type= 0
Boundary for River Rch & Prof#=LtWekiva,LtWekiva        , 5
Up Type= 0
Dn Type= 0
Boundary for River Rch & Prof#=LtWekiva,LtWekiva        , 6
Up Type= 0
Dn Type= 0
Boundary for River Rch & Prof#=LtWekiva,LtWekiva        , 7
Up Type= 0
Dn Type= 0
Boundary for River Rch & Prof#=LtWekiva,LtWekiva        , 8
Up Type= 0
Dn Type= 0
Boundary for River Rch & Prof#=LtWekiva,LtWekiva        , 9
Up Type= 0
Dn Type= 0
Boundary for River Rch & Prof#=LtWekiva,LtWekiva        , 10
Up Type= 0
Dn Type= 0
Boundary for River Rch & Prof#=LtWekiva,LtWekiva        , 11
Up Type= 0
Dn Type= 0
Boundary for River Rch & Prof#=LtWekiva,LtWekiva        , 12
Up Type= 0
Dn Type= 0
Boundary for River Rch & Prof#=LtWekiva,LtWekiva        , 13
Up Type= 0
Dn Type= 0
Boundary for River Rch & Prof#=LtWekiva,LtWekiva        , 14
Up Type= 0
Dn Type= 0
Boundary for River Rch & Prof#=ROK,ROK             , 1
Up Type= 0
Dn Type= 0
Boundary for River Rch & Prof#=ROK,ROK             , 2
Up Type= 0
Dn Type= 0
Boundary for River Rch & Prof#=ROK,ROK             , 3
Up Type= 0
Dn Type= 0
Boundary for River Rch & Prof#=ROK,ROK             , 4
Up Type= 0
Dn Type= 0
Boundary for River Rch & Prof#=ROK,ROK             , 5
Up Type= 0
Dn Type= 0
Boundary for River Rch & Prof#=ROK,ROK             , 6
Up Type= 0
Dn Type= 0
Boundary for River Rch & Prof#=ROK,ROK             , 7
Up Type= 0
Dn Type= 0
Boundary for River Rch & Prof#=ROK,ROK             , 8
Up Type= 0
Dn Type= 0
Boundary for River Rch & Prof#=ROK,ROK             , 9
Up Type= 0
Dn Type= 0
Boundary for River Rch & Prof#=ROK,ROK             , 10
Up Type= 0
Dn Type= 0
Boundary for River Rch & Prof#=ROK,ROK             , 11
Up Type= 0
Dn Type= 0
Boundary for River Rch & Prof#=ROK,ROK             , 12
Up Type= 0
Dn Type= 0
Boundary for River Rch & Prof#=ROK,ROK             , 13
Up Type= 0
Dn Type= 0
Boundary for River Rch & Prof#=ROK,ROK             , 14
Up Type= 0
Dn Type= 0
Boundary for River Rch & Prof#=wekiva,wek_run         , 1
Up Type= 0
Dn Type= 0
Boundary for River Rch & Prof#=wekiva,wek_run         , 2
Up Type= 0
Dn Type= 0
Boundary for River Rch & Prof#=wekiva,wek_run         , 3
Up Type= 0
Dn Type= 0
Boundary for River Rch & Prof#=wekiva,wek_run         , 4
Up Type= 0
Dn Type= 0
Boundary for River Rch & Prof#=wekiva,wek_run         , 5
Up Type= 0
Dn Type= 0
Boundary for River Rch & Prof#=wekiva,wek_run         , 6
Up Type= 0
Dn Type= 0
Boundary for River Rch & Prof#=wekiva,wek_run         , 7
Up Type= 0
Dn Type= 0
Boundary for River Rch & Prof#=wekiva,wek_run         , 8
Up Type= 0
Dn Type= 0
Boundary for River Rch & Prof#=wekiva,wek_run         , 9
Up Type= 0
Dn Type= 0
Boundary for River Rch & Prof#=wekiva,wek_run         , 10
Up Type= 0
Dn Type= 0
Boundary for River Rch & Prof#=wekiva,wek_run         , 11
Up Type= 0
Dn Type= 0
Boundary for River Rch & Prof#=wekiva,wek_run         , 12
Up Type= 0
Dn Type= 0
Boundary for River Rch & Prof#=wekiva,wek_run         , 13
Up Type= 0
Dn Type= 0
Boundary for River Rch & Prof#=wekiva,wek_run         , 14
Up Type= 0
Dn Type= 0
Boundary for River Rch & Prof#=wekiva,wekiva_riv_up   , 1
Up Type= 0
Dn Type= 0
Boundary for River Rch & Prof#=wekiva,wekiva_riv_up   , 2
Up Type= 0
Dn Type= 0
Boundary for River Rch & Prof#=wekiva,wekiva_riv_up   , 3
Up Type= 0
Dn Type= 0
Boundary for River Rch & Prof#=wekiva,wekiva_riv_up   , 4
Up Type= 0
Dn Type= 0
Boundary for River Rch & Prof#=wekiva,wekiva_riv_up   , 5
Up Type= 0
Dn Type= 0
Boundary for River Rch & Prof#=wekiva,wekiva_riv_up   , 6
Up Type= 0
Dn Type= 0
Boundary for River Rch & Prof#=wekiva,wekiva_riv_up   , 7
Up Type= 0
Dn Type= 0
Boundary for River Rch & Prof#=wekiva,wekiva_riv_up   , 8
Up Type= 0
Dn Type= 0
Boundary for River Rch & Prof#=wekiva,wekiva_riv_up   , 9
Up Type= 0
Dn Type= 0
Boundary for River Rch & Prof#=wekiva,wekiva_riv_up   , 10
Up Type= 0
Dn Type= 0
Boundary for River Rch & Prof#=wekiva,wekiva_riv_up   , 11
Up Type= 0
Dn Type= 0
Boundary for River Rch & Prof#=wekiva,wekiva_riv_up   , 12
Up Type= 0
Dn Type= 0
Boundary for River Rch & Prof#=wekiva,wekiva_riv_up   , 13
Up Type= 0
Dn Type= 0
Boundary for River Rch & Prof#=wekiva,wekiva_riv_up   , 14
Up Type= 0
Dn Type= 0
Boundary for River Rch & Prof#=wekiva,wekiva_riv_down , 1
Up Type= 0
Dn Type= 1
Dn Known WS=-0.03
Boundary for River Rch & Prof#=wekiva,wekiva_riv_down , 2
Up Type= 0
Dn Type= 1
Dn Known WS=1.31
Boundary for River Rch & Prof#=wekiva,wekiva_riv_down , 3
Up Type= 0
Dn Type= 1
Dn Known WS=3.17
Boundary for River Rch & Prof#=wekiva,wekiva_riv_down , 4
Up Type= 0
Dn Type= 1
Dn Known WS=3.49
Boundary for River Rch & Prof#=wekiva,wekiva_riv_down , 5
Up Type= 0
Dn Type= 1
Dn Known WS=4.51
Boundary for River Rch & Prof#=wekiva,wekiva_riv_down , 6
Up Type= 0
Dn Type= 1
Dn Known WS=2.22
Boundary for River Rch & Prof#=wekiva,wekiva_riv_down , 7
Up Type= 0
Dn Type= 1
Dn Known WS=3.49
Boundary for River Rch & Prof#=wekiva,wekiva_riv_down , 8
Up Type= 0
Dn Type= 1
Dn Known WS=3.33
Boundary for River Rch & Prof#=wekiva,wekiva_riv_down , 9
Up Type= 0
Dn Type= 1
Dn Known WS=2.93
Boundary for River Rch & Prof#=wekiva,wekiva_riv_down , 10
Up Type= 0
Dn Type= 1
Dn Known WS=1.89
Boundary for River Rch & Prof#=wekiva,wekiva_riv_down , 11
Up Type= 0
Dn Type= 1
Dn Known WS=1.55
Boundary for River Rch & Prof#=wekiva,wekiva_riv_down , 12
Up Type= 0
Dn Type= 1
Dn Known WS=0.91
Boundary for River Rch & Prof#=wekiva,wekiva_riv_down , 13
Up Type= 0
Dn Type= 1
Dn Known WS=0.01
Boundary for River Rch & Prof#=wekiva,wekiva_riv_down , 14
Up Type= 0
Dn Type= 1
Dn Known WS=-0.14
DSS Import GetInterval= 0
DSS Import GetPeak= 0
DSS Import FillOption= 0

--- wekiva_ras.u02 (unsteady flow) ---

Flow Title=unsteady_BC_2009
Program Version=5.03
Use Restart= 0
Boundary Location=LtWekiva        ,LtWekiva        ,312.14  ,        ,                ,                ,                ,
Interval=1DAY
Flow Hydrograph= 182
    5.98    4.97    5.18    5.01    4.97    4.84    4.89    4.63    4.57    7.13
    18.1    11.7    11.2    14.3      14    12.9    11.9      11    10.3    9.75
    9.23    8.71    8.48    8.23    8.07    7.82    7.72    7.78    7.38    6.98
    10.6    8.01    7.48    7.32    6.98    6.81    6.71    6.44    6.69    6.68
    6.82    6.59    6.47    6.32     6.2     6.1     6.2     6.3     6.2     6.4
     6.3     6.5     6.6    6.68    6.83    7.02    7.17    6.99     7.1    7.15
    6.88    7.08    8.84    7.28    7.19    7.52    7.45    7.26    7.83    7.32
    10.1    9.07    8.22    9.13     7.8    7.43    7.36    6.47    5.99    5.28
    5.54    5.03    4.91    4.84     8.3    5.06     4.8    4.96    4.36    4.12
    4.04       4    3.43    3.29    3.14    2.86    2.32    2.11    1.95    1.58
    1.22     1.3    1.08     .75     .81      .8     .87     .58     .37     .32
      .2     .37      .3      .3     .17     .45     .25     .55    38.8     125
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Use DSS=False
Use Fixed Start Time=True
Fixed Start Date/Time=20JAN2009,2400
Is Critical Boundary=False
Boundary Location=ROK             ,ROK             ,480.77  ,        ,                ,                ,                ,
Interval=1DAY
Flow Hydrograph= 182
    55.8    55.6    55.5    55.4    55.4    55.4    55.4    55.6    55.9    56.1
    56.3      56    55.9    56.4    56.4    56.2    56.2    56.2    56.2    56.3
    56.3    56.4    56.4    56.4    56.2    56.1    55.9    55.8    55.7    55.9
    55.9    55.7    55.5    55.2    55.2    55.3    55.3    55.3    55.4    55.5
    55.4    55.1      55    55.1    55.1      55      55    54.8    54.6    54.4
    54.2      54      54    53.8    53.6    53.4    53.5    53.1    53.1      53
    52.8    52.6    52.8    52.8    52.8    52.5    52.3    52.3    52.4    52.3
    52.4    53.3    54.2    53.9    53.7    53.5    53.8    53.9    53.9    53.8
    53.6    53.3    53.3      53    53.4    53.3    53.2    53.1      53    52.8
    52.7    52.6    52.5    52.1      52    51.6    51.3    51.2    51.1    51.1
    51.1    50.8    50.6    50.4    50.1    50.1    50.1    49.8    49.6    49.5
    49.2    48.9    49.2    49.2    49.3    49.3    49.4    49.7      51      53
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Use DSS=False
Use Fixed Start Time=False
Fixed Start Date/Time=01JUN2008,2400
Is Critical Boundary=False
Boundary Location=wekiva          ,wek_run         ,793.32  ,        ,                ,                ,                ,
Interval=1DAY
Flow Hydrograph= 182
    67.3    66.8    66.4    66.4    66.5    66.4    66.3    66.4    66.6    66.5
    66.9    67.1    66.9    67.5    67.4    67.3    66.8    66.8      67      67
    67.1    67.4    67.3    66.9      67    67.1    66.8    66.9    66.7    66.8
      67    66.9    66.5    66.1    65.8    65.9    65.5    65.2    65.2    65.2
    64.8    64.8    64.4    64.1    63.8    63.7    63.6      63    62.9    62.8
    62.4    61.9    62.1    61.6    61.2    61.2    61.2    60.8    60.3    60.3
    59.9    59.6    59.8      60    59.8    59.4    59.5    59.3    58.9      59
    59.2    59.3    59.3    59.2    58.8    58.3    58.4    58.2    57.8    57.3
    57.2    57.1    56.7    56.9    57.3    57.5    57.1      57    56.9    56.7
    56.7      57    56.7    56.2    56.1    55.9    55.6    55.6    55.8    55.5
      55    54.9    54.8    54.5    54.4    54.4    54.2    53.9    53.8    53.6
    53.3    53.2    53.3    53.9      54    54.5    54.5    54.3    54.8    55.2
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Use DSS=False
Use Fixed Start Time=False
Fixed Start Date/Time=01JUN2008,2400
Is Critical Boundary=False
Boundary Location=wekiva          ,wekiva_riv_down ,0       ,        ,                ,                ,                ,
Interval=1HOUR
Stage Hydrograph= 4369
    -.46    -.54    -.54    -.51     -.6    -.66    -.61    -.56    -.53    -.56
    -.55    -.61    -.63    -.62    -.59     -.6     -.6    -.62    -.57    -.52
    -.53    -.54    -.52    -.53    -.52    -.51    -.51    -.51     -.5    -.52
    -.53    -.52    -.53    -.52    -.52    -.53    -.49    -.51    -.51    -.52
    -.51    -.52    -.52    -.51    -.51     -.5     -.5     -.5    -.49    -.49
    -.51    -.49    -.51    -.51    -.51    -.53    -.52    -.52    -.51    -.51
    -.51    -.52    -.51    -.51    -.52    -.53    -.52    -.51    -.52    -.51
    -.53    -.49    -.51    -.52    -.51    -.51    -.52    -.52    -.52    -.53
    -.53    -.52    -.53    -.53    -.52    -.52    -.52    -.53    -.54    -.54
    -.54    -.54    -.54    -.55    -.54    -.53    -.53    -.54    -.54    -.56
    -.55    -.55    -.56    -.56    -.57    -.57    -.56    -.57     -.6    -.58
    -.58    -.59    -.56    -.57    -.56    -.58    -.59    -.57    -.59     -.6
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Use DSS=False
Use Fixed Start Time=True
Fixed Start Date/Time=20JAN2009,0000
Is Critical Boundary=False
Boundary Location=LtWekiva        ,LtWekiva        ,250.47  ,        ,                ,                ,                ,
Interval=1DAY
Lateral Inflow Hydrograph= 182
   43.23      43    42.4   41.61   42.62   42.47   40.74   42.16   42.22   42.91
      46   43.66   43.59   44.77   43.84   44.25   43.84    43.5   43.33      43
   41.72   42.49   42.37   42.16   42.42    42.2   42.31   41.66   42.09      42
   42.67   42.22   42.07   41.91   41.64   41.66   41.67   41.56   41.64   41.43
   41.54   41.27   41.49   41.34   40.95   41.04   41.01   41.13   41.24   41.12
   40.62   40.13   40.62   40.73   40.62   40.96    41.2   40.89   40.19    40.5
   40.17    40.3   40.93   40.92   40.68   40.18   40.88   40.56   40.93   40.53
   40.35   40.51   41.01   41.03   40.79   40.78   40.48   40.58   40.61   39.93
   40.41   40.08   39.98   39.76   41.18   40.15    39.8    39.7   39.89   39.77
   40.36   40.32   40.18   39.48   39.98      40   39.89    40.3   40.41      40
   39.57   39.91   39.38   39.25   37.64   37.47   37.54   37.43   39.12   38.81
   38.59   38.43   39.03   39.39   38.62   39.38   38.96   38.52   43.29   69.47
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Use DSS=False
Use Fixed Start Time=True
Fixed Start Date/Time=20JAN2009,2400
Is Critical Boundary=False
Boundary Location=LtWekiva        ,LtWekiva        ,182.49  ,        ,                ,                ,                ,
Interval=1DAY
Lateral Inflow Hydrograph= 182
    1.42    1.48     1.5    1.45    1.41    1.37    1.33    1.32    1.31    4.52
    9.01     3.2    2.26    4.23    3.43    2.36    2.11    1.92    1.71    1.56
    1.44     1.4    1.35    1.33    1.27    1.22    1.23    1.31    1.24    1.25
    2.23    1.42    1.33    1.23    1.16    1.18     1.2    1.17    1.14     1.1
    1.08     .98    1.13    1.08    1.08    1.03     .97     .95     .92     .89
     .88     .87     .87     .86     .84     .83     .82     .86     .89     .85
     .81     .81     1.2     .95     .83     .78     .78     .76    1.12     .91
     .86    1.71     1.1     .78     .74     .72     .71      .7     .81     .73
     .68     .66     .67     .67     2.4    1.05     .72     .68     .66     .65
    1.35     .86     .67     .64     .61     .59     .58     .61      .6      .6
     .59     .58     .56     .55     .55     .55     .54     .53     .53     .52
     .52     .51     .51    1.97     .91     .54     .52     .79    14.4   56.56
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Use DSS=False
Use Fixed Start Time=False
Is Critical Boundary=False
Boundary Location=LtWekiva        ,LtWekiva        ,143.98  ,30.50   ,                ,                ,                ,
Interval=1DAY
Uniform Lateral Inflow Hydrograph= 182
    3.26    3.42    3.45     3.3    3.22    3.13    3.04    3.05    3.02    9.11
   13.92    6.05    5.23    9.64    6.92    6.25    5.52    4.86    4.15    3.66
    3.33    3.24    3.14     3.1    2.93    2.83    2.87    3.09    2.85    2.93
    4.53    2.75       3    2.73     2.6    2.72    2.77    2.71    2.63    2.55
     2.5    2.25    2.74    2.53    2.55    2.41    2.29    2.26     2.2    2.14
    2.11     2.1    2.11    2.09    2.03    2.03    2.01    2.13    2.18    2.08
    1.97    1.97    2.68    2.17    1.98    1.87    1.91    1.84    2.46    2.04
    2.07    3.53    1.81    1.75    1.71    1.69     1.7    1.67    2.02    1.73
    1.64    1.61    1.64    1.65    4.51    1.83    1.59    1.58    1.57    1.55
    2.85    1.57    1.54    1.51    1.46    1.44    1.42     1.5    1.47    1.46
    1.45    1.41    1.36    1.34    1.35    1.35    1.32    1.31     1.3    1.28
    1.28    1.26    1.25    3.95    1.29    1.28    1.27    2.17      26  147.45
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Use DSS=False
Use Fixed Start Time=False
Is Critical Boundary=False
Boundary Location=ROK             ,ROK             ,350.27  ,        ,                ,                ,                ,
Interval=1DAY
Lateral Inflow Hydrograph= 182
    2.41     2.4    2.42    2.42    2.37    2.31    2.23    2.17    2.11    2.51
    4.42    4.07    3.58    3.57    3.79    3.39    3.12    2.93    2.76    2.59
    2.44    2.32    2.21    2.14    2.06    1.97    1.91    1.94    1.93    1.91
    2.09     2.2    2.09       2    1.88    1.79    1.76    1.73    1.69    1.63
     1.6    1.52    1.48     1.5    1.48    1.44    1.37    1.29    1.22    1.15
    1.08    1.02     .99     .96     .93     .89     .86     .86     .89      .9
     .87     .86    1.05     1.1    1.04     .94     .86     .81     .92       1
     .98    1.15    1.26    1.09     .91     .76     .68     .64     .65     .68
     .62     .53     .48     .48      .9    1.11     .94     .77     .65     .56
     .64     .78     .67     .57     .47     .37     .29     .28      .3     .31
     .31      .3     .25     .19     .15     .14     .12      .1     .09     .07
     .05     .04     .02     .26     .55     .45     .36     .32    2.22     8.9
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Use DSS=False
Use Fixed Start Time=False
Is Critical Boundary=False
Boundary Location=ROK             ,ROK             ,18.17   ,        ,                ,                ,                ,
Interval=1DAY
Lateral Inflow Hydrograph= 182
   15.65   15.57   15.58   15.55   15.44   15.27   15.05   14.83   14.62   15.52
    21.3    22.3    22.1   22.49   23.64      23   22.29   21.56   20.76   19.91
   19.07   18.26   17.52   16.85   16.23    15.6   15.07   14.77   14.48   14.19
   14.45   14.83   14.59   14.36   13.98   13.63   13.39   13.18   12.94   12.68
   12.47   12.17   11.92   11.82   11.68   11.52   11.27      11   10.72   10.43
   10.13    9.86    9.63    9.44    9.24    9.04    8.87    8.77    8.76    8.75
    8.66     8.6    9.03    9.25     9.2    9.01     8.8     8.6    8.78       9
    8.98    9.44    9.98    9.77    9.41    8.95    8.61    8.32    8.14    8.06
    7.81    7.48    7.21    7.04    7.97    8.82     8.7     8.4    8.08    7.74
    7.78    8.14    7.89    7.58    7.21     6.8    6.42    6.17    6.03    5.88
    5.77    5.63    5.42    5.18    4.96    4.81    4.66    4.51    4.37    4.22
    4.07    3.93     3.8    4.47     5.5    5.53    5.46    5.39   10.35   31.14
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Use DSS=False
Use Fixed Start Time=False
Is Critical Boundary=False
Boundary Location=ROK             ,ROK             ,350.27  ,215.81  ,                ,                ,                ,
Interval=1DAY
Uniform Lateral Inflow Hydrograph= 182
   12.51   12.87   12.87    12.4   12.08   11.75   11.41   11.32   11.14   11.75
   13.52   13.58   13.29   13.78   13.71   13.74   13.73   13.61   12.96   12.65
   12.25    12.1   11.86   11.75   11.29      11   11.03   11.53   10.86   10.96
   10.83   10.44   11.03   10.27    9.84   10.03   10.05    9.79    9.49    9.17
    8.95     8.2    9.35    8.73    8.67    8.22    7.82    7.71    7.54    7.37
    7.23    7.22    7.25    7.17    6.93    6.94    6.82    7.21    7.32    7.04
    6.71    6.63    7.18    7.25    6.75    6.32    6.55    6.24    6.17    6.86
    6.44    6.13    6.14    5.91     5.8    5.76    5.78    5.69    6.74    5.93
    5.59    5.51    5.57    5.64    5.88    6.19    5.44     5.4    5.36    5.32
    5.38    5.37    5.28    5.18    5.04    4.99    4.94    5.15    5.05    5.03
       5    4.88    4.75    4.67     4.7     4.7     4.6    4.59    4.54    4.48
    4.46    4.42    4.39    4.84    4.52     4.5    4.46    4.44    6.52   13.91
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Use DSS=False
Use Fixed Start Time=False
Is Critical Boundary=False
Boundary Location=wekiva          ,wekiva_riv_up   ,711.81  ,579.74  ,                ,                ,                ,
Interval=1DAY
Uniform Lateral Inflow Hydrograph= 182
    3.83    4.01    4.04    3.87    3.78    3.67    3.58    3.58    3.54    8.19
   16.48   10.39    8.27   12.33   12.87   11.12    9.09     7.3    5.67    4.47
     3.8    3.69     3.6    3.58    3.42    3.34     3.4    3.65    3.39    3.47
    4.63    3.22    3.51    3.21    3.07    3.21    3.27    3.19    3.11    3.01
    2.96    2.66    3.22    2.99       3    2.85     2.7    2.67     2.6    2.53
    2.49    2.49    2.51    2.48    2.39     2.4    2.36    2.52    2.58    2.46
    2.33    2.32    2.94    2.57    2.35    2.19    2.27    2.17    2.62    2.42
    2.38    3.42    2.13    2.04       2    1.98    1.99    1.96    2.39    2.05
    1.92    1.89    1.92    1.94    4.13    2.17    1.87    1.85    1.84    1.82
     2.8    1.84    1.81    1.76    1.71    1.69    1.67    1.76    1.72    1.71
     1.7    1.65     1.6    1.57    1.58    1.58    1.54    1.54    1.52     1.5
    1.49    1.48    1.47    3.55    1.52    1.51    1.49    2.16   22.85  240.24
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Use DSS=False
Use Fixed Start Time=False
Is Critical Boundary=False
Boundary Location=wekiva          ,wekiva_riv_down ,508.92  ,370.65  ,                ,                ,                ,
Interval=1DAY
Uniform Lateral Inflow Hydrograph= 182
     7.6    7.97    8.02    7.69     7.5     7.3     7.1    7.11    7.04   11.71
   15.93   10.13    9.34   12.83   10.85   10.38    9.82    9.26    8.37    7.82
    7.32    7.13    6.93    6.91    6.61    6.48    6.62    7.13    6.63    6.82
     7.9    6.35    6.93    6.35    6.08    6.35    6.46    6.32    6.14    5.95
    5.85    5.27    6.37     5.9    5.93    5.62    5.34    5.27    5.13       5
    4.91    4.91    4.94    4.89    4.71    4.72    4.64    4.97    5.07    4.84
    4.58    4.55    5.39    5.06    4.64    4.32    4.48    4.27    4.67    4.76
    4.54    5.44    4.19    4.02    3.94     3.9    3.92    3.85     4.7    4.04
    3.78    3.72    3.78    3.83    6.04    4.27    3.67    3.64    3.61    3.58
    4.55    3.63    3.56    3.47    3.36    3.32    3.29    3.47    3.38    3.37
    3.35    3.25    3.15    3.09    3.11    3.11    3.04    3.03    2.99    2.95
    2.94    2.91    2.89    5.08    2.98    2.96    2.94    3.57   22.18  114.69
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Use DSS=False
Use Fixed Start Time=False
Is Critical Boundary=False
Boundary Location=wekiva          ,wekiva_riv_down ,386.11  ,        ,                ,                ,                ,
Interval=1DAY
Lateral Inflow Hydrograph= 182
   18.46   18.38   18.32   18.33    18.3   18.23   18.16   18.19   18.17   18.14
   18.34   18.39   18.41   18.52   18.52   18.51   18.41   18.42   18.38   18.34
   18.31   18.32   18.26    18.2   18.16   18.15   18.09   18.05   18.05   18.04
   18.02   18.01   18.01   17.96   17.93   17.94   17.88   17.84   17.85   17.82
   17.79   17.77   17.77   17.73   17.66   17.62    17.6   17.54   17.56   17.56
    17.5    17.4   17.42   17.37   17.29   17.27   17.28   17.24   17.17   17.16
    17.1   17.03    17.1   17.15   17.11   17.05   17.09   17.06   17.01   17.05
    17.2   17.29   17.32    17.3   17.26   17.21   17.18   17.15    17.1   17.02
   16.97   16.91   16.86   16.88   16.98   17.02   16.98   16.92    16.9   16.84
   16.86   16.89   16.82   16.69   16.66   16.58   16.51   16.47   16.48   16.42
   16.32    16.3   16.27   16.18   16.14   16.14   16.08   15.96   15.93   15.86
   15.76   15.75   15.82   15.98   15.97   16.07   16.04   15.98   16.25   16.86
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Use DSS=False
Use Fixed Start Time=False
Is Critical Boundary=False
Boundary Location=wekiva          ,wekiva_riv_down ,370.65  ,        ,                ,                ,                ,
Interval=1DAY
Lateral Inflow Hydrograph= 182
    1.32     1.3     1.3    1.29    1.27    1.26    1.25    1.23    1.21    1.24
    1.45    1.46    1.44    1.46    1.51    1.49    1.47    1.46    1.44    1.42
    1.39    1.37    1.35    1.33     1.3    1.28    1.26    1.24    1.22    1.21
    1.21    1.21    1.19    1.18    1.16    1.14    1.12     1.1    1.08    1.07
    1.05    1.03    1.01       1     .98     .96     .94     .92      .9     .88
     .86     .84     .82      .8     .78     .76     .74     .73     .71      .7
     .69     .67     .68     .68     .67     .65     .63     .62     .62     .62
     .61     .62     .64     .62      .6     .58     .57     .55     .54     .53
     .51      .5     .48     .47     .49     .52      .5     .49     .47     .45
     .45     .46     .45     .43     .41      .4     .38     .36     .35     .34
     .33     .32      .3     .29     .27     .26     .24     .23     .22      .2
     .19     .17     .16     .18      .2      .2     .19     .18     .36    1.05
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Use DSS=False
Use Fixed Start Time=False
Is Critical Boundary=False
Boundary Location=wekiva          ,wekiva_riv_down ,344.64  ,322.22  ,                ,                ,                ,
Interval=1DAY
Uniform Lateral Inflow Hydrograph= 182
    2.07    2.17    2.18    2.09    2.04    1.99    1.93    1.93    1.92    3.19
    4.34    2.76    2.54    3.49    2.96    2.82    2.67    2.52    2.28    2.13
    1.99    1.94    1.89    1.88     1.8    1.76     1.8    1.94    1.81    1.86
    2.15    1.73    1.89    1.73    1.66    1.73    1.76    1.72    1.67    1.62
    1.59    1.43    1.73    1.61    1.61    1.53    1.45    1.44     1.4    1.36
    1.34    1.34    1.35    1.33    1.28    1.29    1.26    1.35    1.38    1.32
    1.25    1.24    1.47    1.38    1.26    1.18    1.22    1.16    1.27     1.3
    1.24    1.48    1.14     1.1    1.07    1.06    1.07    1.05    1.28     1.1
    1.03    1.01    1.03    1.04    1.64    1.16       1     .99     .98     .98
    1.24     .99     .97     .95     .91      .9      .9     .94     .92     .92
     .91     .88     .86     .84     .85     .85     .83     .82     .82      .8
      .8     .79     .79    1.38     .81     .81      .8     .97    6.04   31.22
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Use DSS=False
Use Fixed Start Time=False
Is Critical Boundary=False
Boundary Location=wekiva          ,wekiva_riv_down ,143.23  ,        ,                ,                ,                ,
Interval=1DAY
Lateral Inflow Hydrograph= 182
     .39     .37     .36     .35     .34     .32     .31     .29     .28     .44
     1.5    1.58     1.5    1.59    1.84    1.74    1.66    1.57    1.49    1.41
    1.33    1.25    1.17     1.1    1.03     .96      .9     .85      .8     .75
     .79     .84     .79     .74     .69     .64      .6     .56     .52     .49
     .45     .42     .39     .36     .33     .31     .28     .25     .22      .2
     .18     .15     .13     .12      .1     .08     .07     .06     .05     .04
     .03     .02     .05     .06     .05     .04     .03     .02     .04     .06
     .05      .1     .18     .16     .13      .1     .08     .06     .05     .04
     .02     .01       0       0     .11     .18     .15     .12      .1     .07
     .09     .14     .11     .09     .06     .04     .02     .01       0       0
       0       0       0       0       0       0       0       0       0       0
       0       0       0       0       0       0       0       0     .81     5.4
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Use DSS=False
Use Fixed Start Time=False
Is Critical Boundary=False
Boundary Location=wekiva          ,wekiva_riv_down ,276.66  ,25.630* ,                ,                ,                ,
Interval=1DAY
Uniform Lateral Inflow Hydrograph= 182
    3.44    3.61    3.63    3.48     3.4    3.31    3.22    3.22    3.19    3.41
    4.93    4.77    4.29    4.63    5.12    4.81    4.46    4.13    3.68    3.41
    3.21    3.18    3.13    3.14    3.01    2.95    3.01    3.24    3.01    3.09
    3.05    2.88    3.14    2.88    2.76    2.88    2.93    2.86    2.79     2.7
    2.66     2.4    2.89    2.68     2.7    2.56    2.44    2.41    2.35    2.29
    2.24    2.24    2.26    2.24    2.15    2.16    2.12    2.28    2.33    2.22
     2.1    2.08    2.29    2.32    2.13    1.98    2.06    1.95    1.93    2.18
    2.02    1.93    1.91    1.84     1.8    1.78    1.79    1.76    2.15    1.85
    1.73     1.7    1.72    1.75    1.85    1.96    1.68    1.66    1.65    1.63
    1.66    1.65    1.62    1.59    1.53    1.52     1.5    1.58    1.55    1.54
    1.53    1.48    1.44    1.41    1.42    1.42    1.39    1.38    1.37    1.35
    1.34    1.33    1.32    1.49    1.36    1.35    1.34    1.34    2.96   45.84
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Use DSS=False
Use Fixed Start Time=False
Is Critical Boundary=False
Boundary Location=wekiva          ,wekiva_riv_down ,25.630* ,        ,                ,                ,                ,
Interval=1DAY
Lateral Inflow Hydrograph= 182
   49.72   49.66   49.58   49.31   49.06    48.9   48.49   48.11   47.97   49.72
   64.16    66.5   64.79   65.39   69.82   68.16   66.27   64.26    62.2   60.15
   58.45   57.16   56.06   55.02   54.06   53.14   52.35   51.74   51.18   50.71
   51.17   51.99   51.47   50.95   50.32   49.76   49.35   48.98   48.61   48.23
   47.93   47.57    47.3   47.17   46.93   46.67   46.38    46.1   45.87   45.64
   45.34   44.98   44.68   44.51   44.33   44.18   44.11   44.06   43.95    43.8
    43.6   43.44   43.91   44.21   44.06   43.75   43.51   43.35   43.65   43.95
   43.74   44.25   45.24   44.76   44.33   43.91   43.59   43.32   43.18   43.04
   42.76   42.47   42.21   42.02   43.63      45   44.41   43.77   43.26   42.85
   43.06    43.8   43.38   42.89   42.42   42.06   41.75   41.62   41.61   41.55
   41.41   41.27   41.08   40.82   40.42   39.95   39.56   39.24   39.19   39.27
   39.25   39.19    39.2   40.47   42.16   41.82   41.51   41.21   50.93  141.36
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Use DSS=False
Use Fixed Start Time=False
Is Critical Boundary=False
Boundary Location=wekiva          ,wekiva_riv_up   ,747.19  ,        ,                ,                ,                ,
Interval=1DAY
Lateral Inflow Hydrograph= 182
    2.26    2.35    2.36    2.26     2.2    2.14    2.08    2.07    2.05    4.74
    5.84    2.43    2.37    4.17    2.43    2.43    2.43    2.41    2.28    2.23
    2.15    2.13    2.09    2.08    1.99    1.94    1.97    2.09    1.95    1.99
    2.68    1.87    2.02    1.85    1.77    1.83    1.85    1.81    1.75    1.69
    1.66     1.5    1.78    1.65    1.65    1.56    1.49    1.47    1.43    1.39
    1.37    1.37    1.38    1.36    1.32    1.32     1.3    1.38    1.41    1.34
    1.27    1.27    1.62     1.4    1.29    1.21    1.24     1.2    1.46    1.32
     1.3    1.93    1.18    1.14    1.11     1.1    1.11    1.09     1.3    1.13
    1.07    1.05    1.07    1.08    2.34    1.19    1.04    1.03    1.02    1.02
    1.58    1.03    1.01     .98     .95     .94     .93     .99     .96     .96
     .95     .92     .89     .88     .88     .88     .87     .86     .85     .84
     .84     .83     .82    2.03     .85     .84     .84    1.22   11.25   21.11
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Use DSS=False
Use Fixed Start Time=False
Is Critical Boundary=False
Observed RC=SR464,LtWekiva        ,LtWekiva        ,312.14  ,0
Observed RC Data= 99
    22.3    5.98   22.24    4.97   22.24    4.89   22.22    4.57   22.76    18.1
   22.56    11.2   22.68      14   22.61    11.9   22.56    10.3   22.53    9.23
    22.5    8.48   22.49    7.82    22.5    7.72   22.51    7.78   22.48    6.98
   22.62    10.6   22.54    8.01   22.52    7.48    22.5    6.81   22.51    6.69
   22.51    6.68   22.52    6.59   22.52     6.2   22.55     6.2   22.57     6.6
   22.58    6.68   22.59    6.83    22.6    7.02   22.61    7.17   22.61    6.99
   22.63    7.15   22.62    6.88   22.63    7.08   22.72    8.84   22.67    7.52
   22.67    7.45    22.7    7.83   22.68    7.32    22.8    10.1   22.77    9.07
   22.74    8.22   22.73     7.8   22.67    6.47   22.63    5.54   22.61    4.91
   22.77     8.3   22.63    5.06   22.63    4.96    22.6    4.36   22.59    4.04
   22.56    3.43   22.55    3.29   22.55    3.14   22.49    2.32   22.48    2.11
   22.46    1.95   22.43    1.58    22.4     1.3   22.37    1.08   22.33     .81
   22.33      .8   22.29     .58   22.26     .37   22.22      .2   22.25     .37
   22.24      .3   22.21     .17   22.28     .45   22.25     .55   23.32    38.8
   24.72     125   25.64     207   26.42     298   26.67     340   26.49     322
   26.16     286   26.16     286   26.29     300    26.1     279   25.85     253
   25.63     231   25.18     189   24.73     151    23.5    65.1   24.02    97.8
   24.62     142   23.56    68.5   23.03    41.2   23.21    50.6   22.98      39
   22.69    27.1   22.74    28.8   24.06     100   24.73     151   23.61    71.4
   23.28    53.1   22.99    39.3   23.16    47.4    23.3    54.3
Observed RC Point Data= 182
            22.3            5.98
           22.24            4.97
           22.25            5.18
           22.24            5.01
           22.24            4.97
           22.23            4.84
           22.24            4.89
           22.22            4.63
           22.22            4.57
           22.34            7.13
           22.76            18.1
           22.57            11.7
           22.56            11.2
           22.67            14.3
           22.68             14.
           22.64            12.9
           22.61            11.9
           22.58             11.
           22.56            10.3
           22.54            9.75
           22.53            9.23
           22.51            8.71
            22.5            8.48
            22.5            8.23
            22.5            8.07
           22.49            7.82
            22.5            7.72
           22.51            7.78
           22.49            7.38
           22.48            6.98
           22.62            10.6
           22.54            8.01
           22.52            7.48
           22.52            7.32
            22.5            6.98
            22.5            6.81
            22.5            6.71
           22.49            6.44
           22.51            6.69
           22.51            6.68
           22.52            6.82
           22.52            6.59
           22.51            6.47
           22.51            6.32
           22.52             6.2
           22.53             6.1
           22.54             6.2
           22.55             6.3
           22.55             6.2
           22.55             6.4
           22.56             6.3
           22.57             6.5
           22.57             6.6
           22.58            6.68
           22.59            6.83
            22.6            7.02
           22.61            7.17
           22.61            6.99
           22.62             7.1
           22.63            7.15
           22.62            6.88
           22.63            7.08
           22.72            8.84
           22.65            7.28
           22.65            7.19
           22.67            7.52
           22.67            7.45
           22.67            7.26
            22.7            7.83
           22.68            7.32
            22.8            10.1
           22.77            9.07
           22.74            8.22
           22.78            9.13
           22.73             7.8
           22.71            7.43
           22.71            7.36
           22.67            6.47
           22.65            5.99
           22.62            5.28
           22.63            5.54
           22.61            5.03
           22.61            4.91
           22.61            4.84
           22.77             8.3
           22.63            5.06
           22.62             4.8
           22.63            4.96
            22.6            4.36
           22.59            4.12
           22.59            4.04
           22.59              4.
           22.56            3.43
           22.55            3.29
           22.55            3.14
           22.53            2.86
           22.49            2.32
           22.48            2.11
           22.46            1.95
           22.43            1.58
           22.39            1.22
            22.4             1.3
           22.37            1.08
           22.33            0.75
           22.33            0.81
           22.33             0.8
           22.33            0.87
           22.29            0.58
           22.26            0.37
           22.25            0.32
           22.22             0.2
           22.25            0.37
           22.25             0.3
           22.24             0.3
           22.21            0.17
           22.28            0.45
           22.24            0.25
           22.25            0.55
           23.32            38.8
           24.72            125.
           25.64            207.
           26.42            298.
           26.67            340.
           26.49            322.
           26.16            286.
           26.16            286.
           26.29            300.
            26.1            279.
           25.85            253.
           25.63            231.
           25.18            189.
           24.73            151.
           24.39            124.
           24.04            99.9
            23.5            65.1
           23.63            76.1
           23.74            79.5
           24.02            97.8
           24.36            122.
           24.75            152.
           24.62            142.
           24.13            105.
           23.88            88.2
           23.56            68.5
            23.3            54.4
           23.12            45.1
           23.03            41.2
           22.99            39.4
           23.16            47.1
           23.21            50.6
           22.98             39.
           22.88            34.5
           22.78            30.3
           22.69            27.1
           22.84            34.6
           22.78            30.5
           22.74            28.8
           23.45            68.8
            24.1            103.
           24.06            100.
           23.85            86.6
           24.16            110.
           24.77            154.
            24.9            165.
           24.73            151.
           24.29            117.
           23.87            87.5
           23.61            71.4
           23.55            67.9
           23.36            57.3
           23.28            53.1
           23.25            51.7
           23.21            49.8
           23.06            42.7
           22.98            38.9
           22.93            36.9
            22.8            31.5
           22.99            39.3
           23.11            45.2
           23.16            47.4
            23.3            54.3
           23.39            59.2
